HEC-RAS study WFKGLADYFK.prj: WFKGLADYFK

--- WFKGLADYFK.g01 (geometry) --- (continued)

Type RM Length L Ch R = 1 ,12320   ,125.1,125.1,125.1
XS GIS Cut Line= 2
2330681.74514936650468.7507616752331360.92028624650283.354305392
#Sta/Elev= 30
       0 2908.99      15  2904.6    27.4 2902.19      73 2895.33    89.6  2888.5
   102.6 2888.09   110.3 2889.31   131.1 2889.76   160.1 2887.99   180.8 2884.43
   203.6  2878.3     214 2871.34   218.1    2870   232.9 2869.64   247.62871.183
   255.7 2872.62   267.9 2871.33     285 2873.15   342.5 2872.68   359.1 2873.83
   469.3 2872.64     525 2873.15   591.5 2875.27     620 2878.01   646.6 2882.11
   665.9 2890.02   686.7 2890.42   690.8 2892.02   699.1 2898.03     704 2899.24
#Mann= 4, -1 ,  0
       0     0.1       0     214   0.045       0   247.6     0.1       0
     620    0.06       0
#XS Ineff= 2 , 0
                          510.02         2881.37
Permanent Ineff=
       F       F
Bank Sta=214,247.6
XS Rating Curve= 0 ,0
Exp/Cntr(USF)=0,0
Exp/Cntr=0.3,0.1

Type RM Length L Ch R = 1 ,12194   ,179.8,179.8,179.8
XS GIS Cut Line= 3
2330616.34281222650628.5091635472331102.70858773650474.843502906
2331415.21762543650364.765168002
#Sta/Elev= 30
       0 2916.37    29.2 2912.18    66.9 2915.88   142.5 2913.72   157.1 2909.74
   180.2  2909.3   222.2 2900.75   247.3 2900.37   285.1 2897.44   297.7 2894.32
   318.6 2879.82   335.82870.457     348  2868.5   364.8 2868.52   372.3 2870.42
   389.9 2871.65   440.3 2871.33   461.3 2872.97   540.7 2871.41   621.9 2872.03
   656.8 2875.63   689.7 2876.36   736.4 2879.66   761.8 2880.47     783  2879.4
   787.3    2880     800 2886.86     817 2887.26   825.4  2885.1   841.4 2887.51
#Mann= 4, -1 ,  0
       0     0.1       0   335.8   0.045       0   372.3     0.1       0
  770.06    0.06       0
Bank Sta=335.8,372.3
XS Rating Curve= 0 ,0
Exp/Cntr(USF)=0,0
Exp/Cntr=0.3,0.1

Type RM Length L Ch R = 1 ,12015   ,366,366,366
XS GIS Cut Line= 3
2330826.03445919650800.8508292382331195.39800041650559.033897578
2331460.13139257650423.920770228
#Sta/Elev= 30
       0 2950.85    43.2 2942.72    53.3 2938.41    64.9 2938.21    74.3 2933.19
     103 2923.98   116.2 2918.22   165.1 2902.61   206.5 2885.35   220.9 2877.32
   236.8 2871.55   251.2 2869.54   285.5 2870.61   294.2 2868.45   303.8 2868.09
   320.7  2870.6   332.4 2871.77   393.7 2870.93   413.7 2868.13   423.3 2869.67
   451.3 2869.96   479.1 2873.83   509.7 2873.21     613 2878.38   639.9 2877.97
   672.4  2883.3   684.9 2888.59   705.1 2889.57     720 2894.81   738.7  2895.3
#Mann= 4, -1 ,  0
       0     0.1       0   285.5   0.045       0   320.7     0.1       0
  621.48    0.06       0
#XS Ineff= 2 , 0
                          485.25         2884.01
Permanent Ineff=
       F       F
Bank Sta=285.5,320.7
XS Rating Curve= 0 ,0
Exp/Cntr(USF)=0,0
Exp/Cntr=0.3,0.1

Type RM Length L Ch R = 1 ,11649   ,285.7,285.7,285.7
XS GIS Cut Line= 2
 2330874.9765044650900.483146453 2331496.9033816650508.581268716
#Sta/Elev= 30
       0 2969.07    43.9 2954.82    53.4 2949.88      70 2947.13    95.5 2933.89
   104.8 2930.76   124.3 2920.76   141.3 2914.91   204.7 2886.25   223.6 2876.89
   235.3 2873.17   247.3 2871.55   281.7 2870.62   313.5 2870.04   337.1 2871.83
   426.7  2870.7   445.8 2868.86   461.5 2867.33   469.5 2867.47   473.72868.963
   478.9 2870.03   516.8 2870.63   611.3 2874.57   639.7 2878.08   651.5 2880.25
   670.3 2885.72   687.7 2892.85   710.6 2894.22   724.8  2903.1   735.1 2906.02
#Mann= 4, -1 ,  0
       0     0.1       0   445.8   0.045       0   473.7     0.1       0
     680    0.06       0
Bank Sta=445.8,473.7
XS Rating Curve= 0 ,0
Exp/Cntr(USF)=0,0
Exp/Cntr=0.3,0.1

Type RM Length L Ch R = 1 ,11363   ,154.4,154.4,154.4
XS GIS Cut Line= 2
 2331030.4407013650988.9855280632331549.58417814650821.855189356
#Sta/Elev= 30
       0  2927.9       6 2923.84    18.6 2920.33    31.2 2910.58    35.4 2908.22
    43.8 2906.99    56.5 2899.52    64.9  2896.2    81.7 2887.23   102.7 2878.75
   112.5 2873.24   119.5 2870.45   141.1 2869.27   185.6 2869.84  197.86 2867.58
   203.5 2866.29   216.1  2866.2   223.7 2867.57   228.7 2868.42   270.8 2869.17
   279.2 2870.48   304.4 2869.32   354.8 2871.38   379.5 2870.33   443.1 2871.03
   451.5 2871.92   464.1 2875.99   506.7 2883.86   514.5 2884.25   545.4 2889.23
#Mann= 3, -1 ,  0
       0     0.1       0  197.86   0.045       0   223.7     0.1       0
Bank Sta=197.86,223.7
XS Rating Curve= 0 ,0
Exp/Cntr=0.3,0.1

Type RM Length L Ch R = 1 ,11209   ,89,89,89
XS GIS Cut Line= 4
2331020.22598724651165.5900358152331211.94509495651067.690916986
2331330.23986353651061.5722220592331613.73939514650888.209199132
#Sta/Elev= 30
       0 2921.42     9.7 2922.73    35.9 2931.93    49.3 2933.82    58.3  2933.3
    80.1 2924.88   107.7  2909.5   116.7  2906.1   141.6 2892.07   170.6 2879.25
   184.1 2870.07   202.4 2867.56   239.5 2868.66   263.9 2867.33   271.6    2866
   291.6 2867.33   299.6 2869.94   364.5 2868.23   500.1 2869.75   518.5  2873.4
   524.5 2875.54   533.3 2876.01   542.3 2878.73   579.8 2884.43   589.2 2887.38
   600.2  2887.8   632.2 2895.08   645.4 2899.81   659.5 2900.04     666    2903
#Mann= 3, -1 ,  0
       0     0.1       0   263.9   0.045       0   291.6     0.1       0
Bank Sta=263.9,291.6
XS Rating Curve= 0 ,0
Exp/Cntr(USF)=0,0
Exp/Cntr=0.3,0.1

Type RM Length L Ch R = 1 ,11120   ,368.8,368.8,368.8
XS GIS Cut Line= 4
2331068.62755264651167.3301208392331183.50882038651172.294126235
2331522.47947455651082.9420291092331608.28585353651031.883687895
#Sta/Elev= 30
       0 2928.19     7.6 2928.01    15.6 2925.54    27.6 2918.34    39.6 2914.77
    62.7 2903.14   103.6 2886.72   132.2 2872.59   152.9 2867.76   165.3 2867.28
     186 2866.56   202.5 2867.31   227.4 2868.67   260.5 2867.72   268.7 2868.56
   310.1 2868.24   318.4 2869.05   330.8 2867.32   343.2 2868.27   359.7  2867.1
   413.5 2868.38   438.3  2871.9   454.9 2875.93   472.2 2877.98   481.5 2879.97
   488.5 2880.16   517.7 2886.73   532.7 2888.75   555.9 2894.77   565.4 2896.14
#Mann= 3, -1 ,  0
       0     0.1       0   165.3   0.045       0   202.5     0.1       0
Bank Sta=165.3,202.5
XS Rating Curve= 0 ,0
Exp/Cntr(USF)=0,0
Exp/Cntr=0.3,0.1

Type RM Length L Ch R = 1 ,10751   ,103.3,103.3,103.3
XS GIS Cut Line= 2
2331237.46264139651383.9395016152331639.61029029651163.567884603
#Sta/Elev= 30
       0    2880    21.3 2875.18    39.4 2873.51    71.5 2873.46    85.2 2872.31
   117.1 2871.48   144.5 2871.82   177.9 2869.41   199.2 2868.71   213.8  2867.3
   235.7 2868.17   249.4    2868  261.35 2866.15   272.2 2864.94     295 2864.87
   299.6 2865.35  301.13 2866.15   308.7 2870.89   313.4 2872.51   319.3 2873.07
   331.5 2873.08   349.7 2875.53   358.9    2878   381.2 2880.49   390.8 2882.38
   399.9 2882.93     409  2884.7   421.9 2884.86   436.4 2886.38   458.6 2887.69
#Mann= 5, -1 ,  0
       0     0.1       0     130    0.06       0     200     0.1       0
  261.35   0.045       0  301.13     0.1       0
Bank Sta=261.35,301.13
XS Rating Curve= 0 ,0
Exp/Cntr=0.3,0.1

Type RM Length L Ch R = 1 ,10647   ,61.5,61.5,61.5
XS GIS Cut Line= 4
2331344.41350956651480.2752038662331418.44810433651399.858316453
2331674.37803966651244.1303757492331772.02711724651217.962975877
#Sta/Elev= 30
       0 2875.84    36.8 2873.58    69.5  2874.2     116 2872.66   120.7 2872.04
     130 2868.69   134.7 2867.93   188.2 2866.65   197.52864.895     205 2863.83
     219 2863.94  224.55 2864.89   228.4 2866.55   242.4 2869.03   268.4 2870.02
   279.9 2873.84   304.6 2876.31   330.8 2880.76   345.4 2881.59   368.7 2884.79
   377.4 2884.77   387.6 2886.53   408.9 2888.36   423.2  2890.9   439.7 2896.39
   464.6 2898.81   478.1 2902.29   487.9 2903.39   501.9 2907.07     510 2907.33
#Mann= 6, -1 ,  0
       0     0.1       0      10    0.06       0   197.5   0.045       0
  224.55    0.06       0  319.31     0.1       0  379.31    0.06       0
Bank Sta=197.5,224.55
XS Rating Curve= 0 ,0
Exp/Cntr(USF)=0,0
Exp/Cntr=0.3,0.1

Type RM Length L Ch R = 1 ,10586   ,135.5,135.5,135.5
XS GIS Cut Line= 4
2331360.40359444651577.0503093082331442.03449325651462.526273454
2331623.27449725651333.0737158712331730.64977622651285.880152333
#Sta/Elev= 30
       0 2876.38     9.7 2875.31      49 2874.91    75.4 2873.67    89.2 2873.74
   107.9 2872.52   127.6  2872.8   132.5 2872.13   143.1 2868.66   149.8 2867.79
   177.4  2868.4   197.3 2866.07   207.2 2865.97   218.7 2864.35   226.3 2864.52
   246.4 2863.84  258.56 2864.54   266.2 2865.98   295.7 2867.21   335.3    2871
   344.8 2872.93   352.5 2875.53     364 2877.13   388.2  2884.1   400.4 2885.19
   412.5 2888.38   421.1 2889.14     452 2894.42   464.8 2898.95   480.7 2901.56
#Mann= 4, -1 ,  0
       0    0.08       0     110    0.06       0   226.3   0.045       0
  258.56    0.06       0
#XS Ineff= 2 , 0
          182.51 2873.67
Permanent Ineff=
       F       F
Bank Sta=226.3,258.56
XS Rating Curve= 0 ,0
Exp/Cntr(USF)=0,0
Exp/Cntr=0.3,0.1

Type RM Length L Ch R = 1 ,10450   ,339.9,339.9,339.9
XS GIS Cut Line= 4
2331436.71922258651910.2517403192331494.69728978651792.069648574
     2331660.938651413.0586187232331718.47657663651309.258922555
#Sta/Elev= 30
       0 2886.49    24.3 2882.94    72.5 2877.92    99.2  2873.9   147.9 2869.89
   200.3 2868.13   238.2 2867.62   287.7 2868.01   331.3 2869.38   374.8  2868.4
   405.2 2866.87   466.8 2867.41   483.9 2865.52   487.42864.342     493 2863.25
   501.7 2863.19     5262864.479   536.6 2865.92   565.5 2865.67   572.8 2866.36
     582 2866.21     586 2867.65   594.9 2872.44   606.6 2880.59   618.5 2885.82
   627.7 2887.86   636.8 2890.76   642.9 2891.86   653.7 2895.48   664.2  2896.4
#Mann= 6, -1 ,  0
       0    0.05       0  261.64    0.07       0  471.64     0.1       0
   487.4   0.045       0     526     0.1       0   575.5    0.06       0
Bank Sta=487.4,526
XS Rating Curve= 0 ,0
Exp/Cntr=0.3,0.1

Type RM Length L Ch R = 1 ,10111   ,182,182,182
XS GIS Cut Line= 2
2331440.18578506 651983.759425032332075.27666224651454.983320241
#Sta/Elev= 30
       0 2890.05    15.6 2885.97    31.2  2883.5    83.3 2878.44   124.9 2867.67
   146.7 2864.83   179.1 2864.31   197.8 2866.81   208.2 2865.28   266.6 2864.71
   499.7 2865.98   566.7 2865.03   586.9 2863.67   591.7 2862.09   603.8 2861.09
   619.4 2862.02   629.8 2864.84   635.2 2868.91   641.7 2875.49   655.8 2885.72
   671.4 2894.49   697.7 2905.05   704.2 2909.41   717.6 2914.77     746 2915.99
   766.7 2930.16     780 2935.13   791.1 2939.31   810.5  2943.7   826.4 2949.29
#Mann= 9, -1 ,  0
       0    0.05       0     140    0.08       0     160    0.07       0
     470    0.05       0   591.7   0.045       0   619.4    0.05       0
     620     0.1       0     650    0.06       0     780     0.1       0
#XS Ineff= 2 , 0
          305.82 2875.83
Permanent Ineff=
       F       F
Bank Sta=591.7,619.4
XS Rating Curve= 0 ,0
Exp/Cntr(USF)=0,0
Exp/Cntr=0.3,0.1

Type RM Length L Ch R = 1 ,9929    ,161.6,161.6,161.6
XS GIS Cut Line= 3
2331468.37970605652026.4936893662331842.22471161651822.069949269
2332152.58220293651686.195683805
#Sta/Elev= 30
       0 2886.37    21.4 2881.76    68.2 2874.87     101 2866.14   118.3 2864.79
   136.5 2865.93   150.2 2864.66   186.7 2864.93   200.4 2863.85   259.6 2865.07
   282.4 2863.78   318.9  2864.7   468.2 2864.74   541.7 2864.08   563.52862.009
   576.7 2860.55   595.3 2862.01   620.3 2863.88   624.7 2865.16   637.8 2875.98
   642.2 2877.61   672.7 2880.51   681.5 2882.32   701.6    2894     712 2901.98
   716.4 2903.72     735 2903.71   751.3 2896.36   755.7 2896.07   764.9 2898.02
#Mann= 7, -1 ,  0
       0    0.05       0      90    0.08       0     200    0.07       0
  536.09     0.1       0   563.5   0.045       0   595.3     0.1       0
  646.09    0.06       0
#XS Ineff= 2 , 0
          259.13 2869.17
Permanent Ineff=
       F       F
Bank Sta=563.5,595.3
XS Rating Curve= 0 ,0
Exp/Cntr=0.3,0.1

Type RM Length L Ch R = 1 ,9767    ,117.7,117.7,117.7
XS GIS Cut Line= 2
2331612.82549154652103.4467981892332180.14039392  651830.8204701
#Sta/Elev= 30
       0 2865.42    22.2 2864.41      57 2864.28    65.8 2863.47    79.1 2865.44
    92.5 2863.66   132.4 2863.25   145.7 2862.36   157.1 2863.68   181.2 2863.94
   225.6  2862.5   375.9 2863.54   423.9 2863.15   435.8 2862.13   460.8 2861.49
   469.7 2860.47   491.9 2859.29  502.26 2860.45   505.2 2861.72   514.1  2867.6
   531.8 2881.57   540.8 2884.76   561.7 2894.18   576.2 2899.29   580.6 2899.36
   585.1 2900.47   597.7 2905.62   607.3 2908.21   616.1  2911.6   629.4 2912.49
#Mann= 7, -1 ,  0
       0    0.05       0      40    0.08       0      60    0.07       0
     370     0.1       0   469.7   0.045       0  502.26     0.1       0
     580    0.06       0
#XS Ineff= 2 , 0
           78.35 2871.46
Permanent Ineff=
       F       F
Bank Sta=469.7,502.26
XS Rating Curve= 0 ,0
Exp/Cntr(USF)=0,0
Exp/Cntr=0.3,0.1

Type RM Length L Ch R = 1 ,9649    ,297,297,297
XS GIS Cut Line= 4
2331603.81642443652172.5698789172332042.64373758652007.445394669
2332082.24542868652004.9900156312332189.05022566651971.507972462
#Sta/Elev= 30
       0 2869.94    60.2 2864.47    74.3 2865.66    85.9 2864.65     150 2863.31
   158.2 2862.56   167.5 2863.66   173.7 2863.63     211 2861.23   226.9 2863.16
   248.3 2862.38   319.7 2862.49   346.6 2861.77   389.3 2862.08   419.6 2863.14
472.83352860.704   486.4 2858.78   502.5 2859.36505.50012860.301   518.9 2862.81
   521.3 2863.93   523.1 2864.87   531.5 2872.25   535.7 2874.86   552.5 2882.08
     561 2886.93   569.3 2888.76   586.5 2895.37   598.6 2897.65   620.5 2904.53
#Mann= 7, -1 ,  0
       0    0.05       0      50    0.08       0     150    0.07       0
  468.87     0.1       0472.8335   0.045       0505.5001     0.1       0
  588.54    0.06       0
#XS Ineff= 2 , 0
          169.76 2870.28
Permanent Ineff=
       F       F
Bank Sta=472.8335,505.5001
XS Rating Curve= 0 ,0
Exp/Cntr(USF)=0,0
Exp/Cntr=0.3,0.1

Type RM Length L Ch R = 1 ,9352    ,138.5,138.5,138.5
XS GIS Cut Line= 3
2331634.21025164652243.9565149312331834.25056195652243.940043083
2332236.69090776652327.773358873
#Sta/Elev= 30
       0 2867.29      10 2866.46      18 2865.42      30  2866.6      46 2865.12
     106 2863.79     178 2863.28   206.1 2863.88   214.3 2863.59   238.8 2861.09
   280.5 2860.04   308.2 2859.94   336.8 2861.49   350.6 2860.51   369.5 2860.99
     390 2860.09   398.1  2860.4   406.3 2859.31   426.7 2859.32   430.8 2859.56
   433.7 2860.41   455.3 2866.75   467.6 2873.27   475.8 2875.77   496.2 2877.53
   508.4 2879.89   545.2 2883.01   573.8 2887.12   598.4 2889.26   611.1  2891.2
#Mann= 6, -1 ,  0
       0    0.05       0      10    0.07       0  210.04    0.08       0
  310.04    0.12       0   398.1   0.045       0   433.7     0.1       0
#XS Ineff= 2 , 0
          209.11 2869.22
Permanent Ineff=
       F       F
Bank Sta=398.1,433.7
XS Rating Curve= 0 ,0
Exp/Cntr=0.3,0.1

Type RM Length L Ch R = 1 ,9214    ,152.8,152.8,152.8
XS GIS Cut Line= 2
2331673.83765201652492.416189054 2332203.0893195652367.313146904
#Sta/Elev= 30
       0 2875.73    24.6 2873.09    84.4 2864.09   125.7 2863.64   149.5 2862.44
   222.7 2861.22   257.5 2860.94   289.4 2861.52   310.7 2860.88323.50522858.335
   331.2 2857.29   339.4 2857.55342.17142858.538   347.7 2859.93   359.4 2860.33
   372.3 2859.82   384.7 2860.32     397 2859.47   410.2 2860.36   416.9 2862.17
   429.9 2869.67   438.1  2872.5   458.6  2875.3   466.9 2875.76   475.1  2877.3
   483.3 2877.85   495.6 2880.11   526.6  2883.1   536.7 2885.31   543.8 2886.01
#Mann= 6, -1 ,  0
       0    0.05       0      70     0.1       0     180    0.12       0
323.5052   0.045       0342.1714    0.12       0     480     0.1       0
Bank Sta=323.5052,342.1714
XS Rating Curve= 0 ,0
Exp/Cntr(USF)=0,0
Exp/Cntr=0.3,0.1

Type RM Length L Ch R = 1 ,9061    ,199.9,199.9,199.9
XS GIS Cut Line= 3
2331677.45362757652616.643420605 2331858.1889582652625.526106224
2332245.16301134652480.721779358
#Sta/Elev= 30
       0 2877.74    27.6 2875.25    62.8 2870.29      95 2867.61   111.8 2863.73
   126.9 2861.76   162.9 2861.19   174.9  2861.5   178.9 2861.03   204.4 2860.72
   307.5 2860.84   332.6 2860.17   364.6 2860.83   369.2 2860.33   375.5 2858.88
   400.9 2859.01  407.54 2857.82   413.7 2856.37     418 2856.27   425.2 2857.81
   435.1 2860.12   443.8 2864.89   456.3 2866.07   467.3 2869.93   477.8 2872.79
   507.7 2875.46   550.4 2880.59   558.9 2883.01   571.3 2883.75   594.1 2886.51
#Mann= 5, -1 ,  0
       0     0.1       0  270.95    0.07       0  340.95     0.1       0
  407.54   0.045       0   425.2     0.1       0
#XS Ineff= 2 , 0
                          532.97         2865.77
Permanent Ineff=
       F       F
Bank Sta=407.54,425.2
XS Rating Curve= 0 ,0
Exp/Cntr=0.3,0.1

Type RM Length L Ch R = 1 ,8861    ,92.8,92.8,92.8
XS GIS Cut Line= 2
2331866.10541633652874.5247684092332300.84604417652563.481059546
#Sta/Elev= 30
       0 2874.17    22.2 2872.12    39.7 2869.68    61.6 2867.65    85.6 2866.34
   108.5 2863.22   131.5 2861.09   171.6 2859.81   238.6 2859.68   242.9 2857.16
   248.5 2855.64   254.7 2855.46   263.4 2855.58   270.4 2857.13   273.1 2857.65
   292.7 2858.89   332.2 2858.37   366.1 2859.53     378 2858.93   394.1 2860.68
   412.4 2859.72   440.3 2859.85     444 2860.59   449.7 2863.44     455    2865
   464.9 2866.08   483.5 2873.85   504.1 2879.79   515.7 2881.56   534.6 2885.99
#Mann= 5, -1 ,  0
       0    0.05       0     210    0.07       0   242.9   0.045       0
   270.4    0.07       0     340     0.1       0
Bank Sta=242.9,270.4
XS Rating Curve= 0 ,0
Exp/Cntr(USF)=0,0
Exp/Cntr=0.3,0.1

Type RM Length L Ch R = 1 ,8768    ,163.7,163.7,163.7
XS GIS Cut Line= 2
2331896.12954377652992.716193559 2332382.3022747652590.182345119
#Sta/Elev= 30
       0 2875.72    31.2 2875.61    57.2 2874.44   130.4 2866.41   150.3 2862.82
     161 2859.77     200 2858.83   241.2 2857.98   280.5  2859.3   287.8 2856.83
   296.1 2855.36   306.5 2855.44   311.6 2856.78   317.9 2858.01     352 2857.29
     369 2858.68   414.5 2858.33   425.8 2860.27   446.7 2860.97   467.4 2859.95
   505.4 2860.72   516.8 2862.78   526.1 2866.23   538.7 2867.29     548 2870.46
   562.2 2874.06   582.6 2876.71   612.8  2884.3   623.2 2887.76   631.2 2889.32
#Mann= 4, -1 ,  0
       0    0.05       0     200    0.07       0   287.8   0.045       0
   311.6     0.1       0
Bank Sta=287.8,311.6
XS Rating Curve= 0 ,0
Exp/Cntr(USF)=0,0
Exp/Cntr=0.3,0.1

Type RM Length L Ch R = 1 ,8605    ,455.9,455.9,455.9
XS GIS Cut Line= 2
 2332035.3507395653079.8427390242332434.31858972 652684.99785609
#Sta/Elev= 30
       0 2872.84    15.2 2872.36    43.6 2869.62    70.3 2868.31    85.6 2866.59
    95.8 2864.41   108.1  2863.2   117.5 2861.44   128.9 2858.41   155.2 2856.93
     170  2856.6     175  2856.9   186.9 2856.54   203.3 2857.41   228.7 2857.68
     257 2857.09   299.5 2858.34   310.9 2857.08   316.4 2856.07   327.7 2855.88
   339.1 2857.06   361.3 2858.52   423.2 2859.54   474.8 2861.32   492.8 2863.46
   507.7 2864.23   517.2  2865.5   528.6 2865.44   541.4 2868.02   561.3 2870.71
#Mann= 5, -1 ,  0
       0    0.06       0     170    0.07       0     280     0.1       0
   310.9   0.045       0   339.1     0.1       0
Bank Sta=310.9,339.1
XS Rating Curve= 0 ,0
Exp/Cntr(USF)=0,0
Exp/Cntr=0.3,0.1

Type RM Length L Ch R = 1 ,8149    ,189.2,189.2,189.2
XS GIS Cut Line= 2
2332085.12334369 653261.67095397 2332654.1871517652831.096125784
#Sta/Elev= 30
       0 2875.29    74.1 2871.17      87 2869.43   104.1 2865.81   124.2 2863.76
   153.3 2863.12     191 2861.09   252.7 2859.13   285.9 2858.72   308.1 2857.37
     319 2857.91   373.7 2858.07   398.6 2856.81   431.7 2857.39   470.3  2856.1
   485.4 2856.71   490.4 2855.99   495.4 2855.27   510.4 2854.85   525.5 2855.94
   559.3  2861.9   577.6  2863.6   587.9 2867.33   617.3 2868.91   655.9 2874.24
   667.8 2876.98   676.4 2877.54   683.6 2878.95   703.5  2879.9   713.6 2881.36
#Mann= 6, -1 ,  0
       0    0.05       0     170    0.06       0     190    0.08       0
     310    0.06       0   490.4   0.045       0   525.5     0.1       0
Bank Sta=490.4,525.5
XS Rating Curve= 0 ,0
Exp/Cntr(USF)=0,0
Exp/Cntr=0.3,0.1

Type RM Length L Ch R = 1 ,7959    ,179.7,179.7,179.7
XS GIS Cut Line= 2
     2332101.005       653437.522332742.37458691653007.957984777
#Sta/Elev= 30
       0 2874.21    29.4 2872.57    71.7 2867.81   119.4 2866.91   152.5 2861.85
   196.4 2858.99   201.5 2859.63   210.8 2858.24   220.5 2859.25   234.9 2858.01
   299.5 2856.13   325.5 2856.72   340.8 2854.64   377.3 2856.64   458.1 2855.98
   523.8 2856.71   576.3 2856.53   582.1  2855.7   584.9  2854.3   590.7 2852.33
   610.4 2852.18   619.5 2852.36   627.42854.188   639.3 2858.76   663.4 2860.65
   697.9 2868.62   721.1 2869.87   726.6 2871.01   743.5 2878.08   771.9 2881.96
#Mann= 6, -1 ,  0
       0    0.05       0     280    0.07       0     500    0.08       0
     520    0.06       0   584.9   0.045       0   627.4    0.06       0
Bank Sta=584.9,627.4
XS Rating Curve= 0 ,0
Exp/Cntr=0.3,0.1

Type RM Length L Ch R = 1 ,7780    ,237.3,237.3,237.3
XS GIS Cut Line= 3
2332309.64292546653519.7299198792332550.25004192653307.100375097
2332852.40781609653172.808031023
#Sta/Elev= 30
       0 2869.05    51.4 2865.39    70.3 2863.33    85.8 2857.92     100 2856.54
   168.9 2855.23   195.6 2855.73   216.9 2855.31   248.9 2853.38   311.9 2855.37
   345.1 2854.19   384.6 2855.59   393.2 2855.04     402 2853.46   410.7 2851.99
   415.1  2851.9   428.3 2852.32   432.6 2853.46     437  2854.7   441.4 2854.94
   454.5 2854.69   475.5 2856.12   493.3 2856.28   515.8 2857.58   541.7 2861.68
   577.1 2863.69     599 2866.35   616.5 2870.38   629.6 2871.45   651.8  2874.5
#Mann= 8, -1 ,  0
       0    0.05       0      30    0.08       0     100    0.05       0
     170    0.07       0     402   0.045       0   432.6    0.12       0
   441.1    0.05       0   521.1    0.12       0
#XS Ineff= 2 , 0
          131.33 2860.16
Permanent Ineff=
       F       F
Bank Sta=402,432.6
XS Rating Curve= 0 ,0
Exp/Cntr(USF)=0,0
Exp/Cntr=0.3,0.1

Type RM Length L Ch R = 1 ,7542    ,312.9,312.9,312.9
XS GIS Cut Line= 2
2332425.54189446653603.9298624572332863.72776619653216.418370537
#Sta/Elev= 30
       0  2865.4    14.2 2864.43      18 2863.94    28.3  2861.5    51.6 2859.34
    67.6 2858.52    83.2 2858.58     137 2856.12     143 2856.36   161.1  2855.9
   168.2 2855.48   173.8 2854.21   179.3 2853.85   196.5 2852.87   207.8 2853.82
   230.5 2854.35   245.7  2853.4   264.5 2854.34   297.2 2854.89   332.5 2854.52
   345.3 2855.17   366.5 2854.81     443 2856.15   477.1 2857.39   489.4 2858.33
   505.5 2860.14   532.2  2864.7   562.1 2871.57   576.2 2871.75     585 2874.49
#Mann= 6, -1 ,  0
       0     0.1       0      10    0.12       0     140     0.1       0
   179.3   0.045       0   207.8     0.1       0     230    0.12       0
Bank Sta=179.3,207.8
XS Rating Curve= 0 ,0
Exp/Cntr=0.3,0.1

Type RM Length L Ch R = 1 ,7230    ,75.4,75.4,75.4
XS GIS Cut Line= 2
2332483.10386989653754.7415220082333059.44184653653480.561319525
#Sta/Elev= 30
       0 2873.25      10 2872.19      59 2867.51      68 2865.08    85.3 2857.52
   103.1 2855.64   187.2 2854.63   206.1 2853.43     329 2854.19   359.2 2852.48
   377.2 2853.82   389.2 2852.26   395.4 2851.12     413  2850.5     422 2850.51
   431.2 2852.22   439.7 2852.83   458.2 2851.31   475.1 2852.92   501.7 2863.32
   510.6 2865.78   527.3 2869.42   537.2 2870.53     546 2872.95   562.3 2875.23
     577 2879.48   590.3 2880.12   594.7 2882.49   608.9 2885.17   638.2 2892.63
#Mann= 9, -1 ,  0
       0    0.05       0      10     0.1       0      60    0.12       0
     160    0.08       0     240    0.12       0     270     0.1       0
   389.2   0.045       0   431.2     0.1       0     600    0.06       0
#XS Ineff= 2 , 0
          136.12 2864.57
Permanent Ineff=
       F       F
Bank Sta=389.2,431.2
XS Rating Curve= 0 ,0
Exp/Cntr(USF)=0,0
Exp/Cntr=0.3,0.1

Type RM Length L Ch R = 1 ,7154    ,373.7,373.7,373.7
XS GIS Cut Line= 3
 2332470.4328164653791.1112812912332922.62255808653632.793939318
 2333054.1224153653616.833185293
#Sta/Elev= 30
       0 2874.33    53.1 2870.84    73.9 2864.67    78.5 2862.09    95.1 2863.21
   107.8 2858.87   124.7 2857.37   188.3 2854.32   260.4 2853.65   269.7 2852.43
   296.4 2853.27   356.9 2852.65   370.6 2853.82   391.7 2852.67   425.7 2852.92
   429.9 2852.54  431.75 2851.37   434.1 2850.08   438.4 2849.85   451.8 2851.36
   459.6 2853.43   473.7 2859.41   480.7 2861.36   500.8 2865.37   512.9 2866.44
     533  2869.9   549.2 2874.31   573.3 2879.18   589.5 2880.72   611.6 2884.82
#Mann= 8, -1 ,  0
       0    0.05       0     120    0.12       0     170    0.08       0
     280    0.12       0     420     0.1       0  431.75   0.045       0
   451.8     0.1       0   579.1    0.06       0
Bank Sta=431.75,451.8
XS Rating Curve= 0 ,0
Exp/Cntr=0.3,0.1

Type RM Length L Ch R = 1 ,6780    ,367.9,367.9,367.9
XS GIS Cut Line= 3
2332564.03974694654101.9099154022332841.42058362653889.795157938
2333139.19707006653800.054299011
#Sta/Elev= 30
       0 2882.57    14.4 2884.28    23.4 2886.06    50.5 2885.73    55.6 2885.36
    67.1 2882.92    85.8 2880.06    90.8 2878.41     116 2864.42   126.1 2860.69
   134.7 2855.79   146.1 2853.82   234.6  2852.2   251.9 2852.94     266 2851.32
   274.5 2849.95   292.2 2851.31   302.3 2851.87   352.1 2852.01   367.9  2852.7
   389.7  2852.2   448.2 2852.87   476.1 2854.76   489.9 2856.75   498.3 2858.59
   527.5  2868.7   565.1 2877.76   602.7 2883.99   644.5 2889.12   660.2 2890.46
#Mann= 7, -1 ,  0
       0    0.08       0     266   0.045       0   292.2    0.08       0
     330     0.1       0  439.19    0.12       0  489.19     0.1       0
  539.19    0.12       0
Bank Sta=266,292.2
XS Rating Curve= 0 ,0
Exp/Cntr(USF)=0,0
Exp/Cntr=0.3,0.1

Type RM Length L Ch R = 1 ,6413    ,305.2,305.2,305.2
XS GIS Cut Line= 3
2332629.55075033654331.5377212432332998.23461872654121.175238622
2333243.92228484653947.551001412
#Sta/Elev= 30
       0 2876.83    12.4 2875.74    30.7 2876.01    72.1 2880.01    95.1 2878.91
   103.3 2875.92   113.5 2874.24   150.4 2857.81   164.2 2855.05   173.4 2855.47
   182.5 2852.05   190.4 2853.24   224.1 2853.23   237.9 2854.37   273.4 2852.02
     376 2850.91   461.1 2851.49   500.3 2850.85   509.1 2849.03   514.8 2847.83
   524.8 2847.65   529.7 2847.72   534.9 2849.02   546.4 2855.68     555 2858.41
     564 2862.94   589.4 2865.39   606.7 2865.55   635.4 2869.48   725.3 2877.93
#Mann= 8, -1 ,  0
       0    0.05       0     120    0.08       0     380     0.1       0
   509.1   0.045       0   534.9     0.1       0  554.48    0.12       0
  574.48     0.1       0  694.48    0.06       0
#XS Ineff= 2 , 0
          236.07 2861.15
Permanent Ineff=
       F       F
Bank Sta=509.1,534.9
XS Rating Curve= 0 ,0
Exp/Cntr=0.3,0.1

Type RM Length L Ch R = 1 ,6107    ,478.8,478.8,478.8
XS GIS Cut Line= 2
2332857.94009625654563.8637662622333441.25567928  654192.6629407
#Sta/Elev= 30
       0 2872.89    45.3 2864.13   140.1 2856.22   157.1 2851.62   163.9 2850.77
   173.3 2851.49   183.8 2847.68   230.2 2850.35   243.4 2848.89   288.1 2850.43
   325.4 2848.83   381.9 2850.36   403.4 2848.82   415.1 2847.09   429.4 2847.49
   433.52848.722   453.1 2851.31     472 2849.18   505.2 2851.27   519.1 2852.45
   541.4 2856.67   557.4 2854.32   581.1 2854.67   590.6 2856.37     600 2860.61
   609.5 2862.17   614.9 2861.53   623.8 2858.33   656.9 2864.97   691.4 2875.42
#Mann= 8, -1 ,  0
       0    0.05       0      80    0.08       0     230     0.1       0
   403.4   0.045       0   433.5    0.12       0     550     0.1       0
     600    0.12       0     660    0.06       0
Bank Sta=403.4,433.5
XS Rating Curve= 0 ,0
Exp/Cntr(USF)=0,0
Exp/Cntr=0.3,0.1

Type RM Length L Ch R = 1 ,5629    ,99.3,99.3,99.3
XS GIS Cut Line= 2
2333022.25797025654821.6043476252333553.83183221 654258.94429491
#Sta/Elev= 30
       0 2904.04    14.4 2905.69    33.6  2905.7    66.9 2900.33    89.4 2891.94
    99.6 2886.69     112 2885.22   117.7 2883.24   127.1 2877.04   138.2  2872.6
   151.6 2864.04   168.6 2857.63   188.4 2847.16   193.2 2845.73   204.2 2845.57
   215.2  2845.7   220.7 2847.07   247.4 2849.74   352.8 2848.78   369.3 2849.93
   468.8  2849.8   550.6 2851.62   584.5 2855.07   600.4 2858.31   638.3 2862.12
   677.4 2863.93   694.9 2871.07   748.7 2884.91     760 2890.41   774.1 2891.17
#Mann= 6, -1 ,  0
       0    0.05       0     150     0.1       0   188.4   0.045       0
   220.7     0.1       0     660    0.12       0     720    0.06       0
Bank Sta=188.4,220.7
XS Rating Curve= 0 ,0
Exp/Cntr(USF)=0,0
Exp/Cntr=0.3,0.1

Type RM Length L Ch R = 1 ,5529    ,265.8,265.8,265.8
XS GIS Cut Line= 2
2333117.89350761 654871.92941888 2333519.0929659654421.168475503
#Sta/Elev= 30
       0 2902.78    20.6 2899.77    48.9  2893.7    57.2 2890.09    74.4 2884.06
    82.9 2881.86    91.4 2878.11   100.1 2875.62   135.8    2861   176.4 2847.18
   182.1 2845.75   189.9 2845.49   199.1 2845.67  211.69 2847.15   233.9 2849.04
   269.9    2849   292.2 2847.98   298.2 2848.75     335 2848.79     416  2847.6
   480.3 2852.11   490.9 2854.34   508.8 2856.15   523.1 2856.75   549.9 2859.81
   561.7 2860.08   571.3 2861.13   581.5 2859.93     593 2864.57   603.4 2866.31
#Mann= 4, -1 ,  0
       0    0.05       0      50     0.1       0   176.4   0.045       0
  211.69     0.1       0
Bank Sta=176.4,211.69
XS Rating Curve= 0 ,0
Exp/Cntr=0.3,0.1

Type RM Length L Ch R = 1 ,5264    ,322.3,322.3,322.3
XS GIS Cut Line= 2
2333276.92396262654967.0229827452333583.52449437654547.384323168
#Sta/Elev= 30
       0 2909.75    49.4 2893.57    59.8 2891.01    73.3 2886.14   106.3 2872.99
     114 2867.41   123.9 2865.06   135.3 2861.05     141 2858.27   149.6 2852.88
   152.5 2852.01   170.7 2849.11   205.4 2848.16   242.8 2849.74   261.3 2847.96
   274.7 2847.59   299.5  2849.1   324.2 2848.25   335.7 2846.58   339.1  2845.4
   349.1 2845.05   364.9 2845.24  370.97 2846.58   384.4 2851.49   413.5 2854.76
   425.9 2855.47   450.2 2857.92   493.7 2863.97   507.4 2867.07   519.7 2868.51
#Mann= 6, -1 ,  0
       0    0.05       0      50     0.1       0   335.7   0.045       0
  370.97     0.1       0     400    0.06       0     410     0.1       0
Bank Sta=335.7,370.97
XS Rating Curve= 0 ,0
Exp/Cntr(USF)=0,0
Exp/Cntr=0.3,0.1

Type RM Length L Ch R = 1 ,4941    ,290.7,290.7,290.7
XS GIS Cut Line= 2
2333591.04127823655073.5030354722333767.72637097654623.938219333
#Sta/Elev= 30
       0 2883.24     4.6 2882.27    17.5 2877.42    30.4 2873.61    51.9 2863.87
    64.8 2860.46      82  2853.4    90.6 2849.03    99.2 2848.34   107.8 2846.63
   122.22845.637   127.6 2844.17   137.9  2843.8   146.5 2843.86   152.3 2845.62
   155.4 2847.08   178.1 2847.49   245.3 2847.89   260.3 2846.22   271.1 2847.45
     353 2848.41   361.4 2849.01     370 2851.66   378.6 2852.71   382.9 2854.14
   391.5 2859.07   404.3 2864.55   430.1 2872.25   447.3 2876.81     483 2884.76
#Mann= 4, -1 ,  0
       0     0.1       0   122.2   0.045       0   152.3     0.1       0
     470    0.06       0
Bank Sta=122.2,152.3
XS Rating Curve= 0 ,0
Exp/Cntr=0.3,0.1

Type RM Length L Ch R = 1 ,4651    ,128,128,128
XS GIS Cut Line= 3
2333681.57869148 655135.651554072333799.99698359655059.496899664
2333972.15225598654623.568785739
#Sta/Elev= 30
       0 2891.71     7.8  2890.8    26.9 2884.89    47.1  2882.2      76 2876.01
    93.7 2871.49   122.9 2861.91   141.3 2858.34   164.8 2851.36     182 2848.61
   195.1 2847.59   251.2 2846.68   358.3 2847.15370.57042845.015     377 2843.53
   388.4 2843.23     397 2843.34404.16962844.748   427.1 2848.45   431.4 2850.04
   441.8 2857.32   478.9 2875.36   500.4 2888.38   513.1 2897.56   521.7  2899.4
   543.2  2898.8   547.5 2899.82     569 2916.31   581.9 2923.59   609.5 2933.75
#Mann= 6, -1 ,  0
       0     0.1       0370.5704   0.045       0404.1696    0.06       0
  430.79     0.1       0  490.79    0.06       0  600.79     0.1       0
Bank Sta=370.5704,404.1696
XS Rating Curve= 0 ,0
Exp/Cntr(USF)=0,0
Exp/Cntr=0.3,0.1

Type RM Length L Ch R = 1 ,4523    ,295.4,295.4,295.4
XS GIS Cut Line= 2
2333828.79425099655206.306933916 2334085.2365154654729.047476566
#Sta/Elev= 30
       0 2896.03    14.9 2891.89      24 2890.35    33.1 2887.07    44.7 2885.16
    65.4  2877.8    77.2 2875.53    91.9 2870.39   101.2 2868.17   112.2 2863.74
   142.2 2856.42   150.8 2852.91   156.9 2848.57   160.2 2847.02   282.8 2846.32
   341.8 2847.62   351.9 2844.88   372.5 2846.02   377.2 2844.68   381.4  2843.3
   387.3 2843.03   400.9 2843.39  406.04  2844.7   419.8 2847.82   467.1 2869.62
   478.9 2876.86   496.6 2890.11   514.6 2891.69   531.1 2890.66   541.8 2895.29
#Mann= 4, -1 ,  0
       0     0.1       0   377.2   0.045       0  406.04     0.1       0
     430    0.06       0
Bank Sta=377.2,406.04
XS Rating Curve= 0 ,0
Exp/Cntr=0.3,0.1

Type RM Length L Ch R = 1 ,4227    ,261.3,261.3,261.3
XS GIS Cut Line= 2
2333879.51886155655212.0718250382334404.53008323655035.916744077
#Sta/Elev= 30
       0 2888.38    51.3 2877.42    76.6 2873.28    97.7 2870.39   127.3 2868.52
   173.7 2862.81   186.3  2859.9   207.4 2852.47   235.4 2844.79   258.1 2843.06
     265 2844.62   274.5 2846.27   279.2 2846.21   287.6 2844.24   300.3 2846.06
   350.9 2845.85   355.1 2846.19   367.8 2850.01   385.1 2851.37   401.5 2854.88
   418.4 2860.39   424.1  2863.7   435.3 2872.03   438.8 2873.46   456.4 2874.01
   464.8 2876.42   477.5  2878.6     507 2891.36   527.2 2898.73   553.8 2911.44
#Mann= 5, -1 ,  0
       0     0.1       0   235.4   0.045       0     265     0.1       0
     340    0.06       0     550     0.1       0
Bank Sta=235.4,265
XS Rating Curve= 0 ,0
Exp/Cntr(USF)=0,0
Exp/Cntr=0.3,0.1

Type RM Length L Ch R = 1 ,3966    ,313.8,313.8,313.8
XS GIS Cut Line= 2
2333882.62133708655316.7495704992334457.66670414655334.775457749
#Sta/Elev= 30
       0  2870.2    29.6 2866.05    65.6  2862.3   117.6 2857.32   177.6 2854.14
   221.7 2848.69   250.3  2848.3   273.5 2849.21   293.7 2845.42   313.7 2846.05
   325.7 2844.91   345.7 2845.88   357.7 2844.68   365.7 2845.05     373 2843.34
   393.7 2842.64   397.8 2843.38   405.8 2850.21   413.8 2852.28     435 2862.47
   449.8 2866.88   465.8 2873.59   477.8 2880.32   489.8 2881.61   501.8 2881.74
   505.8 2883.76   525.8 2899.63   533.5 2904.44   549.8 2910.24   575.3 2921.12
#Mann= 4, -1 ,  0
       0     0.1       0     373   0.045       0   397.8     0.1       0
     420    0.06       0
#XS Ineff= 2 , 0
          273.71 2862.36
Permanent Ineff=
       F       F
Bank Sta=373,397.8
XS Rating Curve= 0 ,0
Exp/Cntr=0.3,0.1

Type RM Length L Ch R = 1 ,3652    ,191.8,191.8,191.8
XS GIS Cut Line= 2
2333699.61962161655467.4448821132334397.33190306655695.410281003
#Sta/Elev= 30
       0 2868.53    62.1 2860.31   118.4 2856.23   150.9 2849.45   168.9  2847.9
   269.9 2847.23   301.8 2848.92   320.4 2847.22   366.7 2846.89   387.7 2848.01
   425.6 2846.56     434 2845.33   439.5 2843.21   446.6 2840.79   452.2 2840.56
   459.3 2841.05   464.9 2843.27   480.8 2843.42   522.4 2850.23   547.4 2851.88
   589.7 2857.89   617.1 2867.38   627.6 2869.99   640.2 2875.97     657 2886.65
   661.3 2888.34   682.3 2888.58   686.5  2889.7   703.3 2900.27     734 2911.06
#Mann= 4, -1 ,  0
       0     0.1       0   439.5   0.045       0   464.9     0.1       0
     640    0.06       0
Bank Sta=439.5,464.9
XS Rating Curve= 0 ,0
Exp/Cntr(USF)=0,0
Exp/Cntr=0.3,0.1

Type RM Length L Ch R = 1 ,3460    ,416.5,416.5,416.5
XS GIS Cut Line= 3
2333501.44885758655578.8862860172334047.79966635655772.726237916
2334375.21638057655912.093522992
#Sta/Elev= 30
       0 2886.43    19.9 2879.92    32.6 2877.33    79.1 2864.72      92 2862.46
   107.3 2860.51   159.9 2856.11     242 2846.81   317.9 2843.48   404.9 2843.41
     457  2844.3     491 2843.76   505.2 2844.66   571.6 2845.67   606.2 2842.93
   619.3 2841.11   631.9 2840.84   636.6 2841.63   639.7 2843.19   645.3 2845.32
     654 2846.08   680.1 2845.71   723.7 2847.53   797.5 2856.04   849.7 2865.98
   875.7 2871.85   884.4  2874.7   914.9  2876.9   927.9 2881.64   935.6 2882.49
#Mann= 5, -1 ,  0
       0    0.05       0      20     0.1       0   606.2   0.045       0
   639.7     0.1       0  859.72    0.06       0
Bank Sta=606.2,639.7
XS Rating Curve= 0 ,0
Exp/Cntr=0.3,0.1

Type RM Length L Ch R = 1 ,3044    ,232.4,232.4,232.4
XS GIS Cut Line= 3
2333451.00127737  655766.9339041 2333862.6263714655865.933458881
2334322.66158256656038.163390156
#Sta/Elev= 30
       0 2860.61    17.7 2859.44    46.5    2856   105.6 2853.19     174 2848.33
   252.2 2845.59     281 2841.77   285.1 2840.53   293.3 2839.95   301.5 2840.25
   311.3 2841.72   350.9 2843.81   371.5 2849.56   375.6  2849.2   396.2 2844.14
   416.7 2843.59   536.1 2845.56   558.1 2847.63   659.9 2845.72     724 2845.68
   762.7 2846.76   784.5 2848.06   809.4 2854.53     818  2855.7   847.9 2855.86
   869.2 2853.98     882 2854.61   894.8 2856.89   903.4 2861.54   914.6 2862.92
#Mann= 10, -1 ,  0
       0    0.05       0     170    0.07       0     230    0.05       0
     281   0.045       0   311.3    0.05       0     370    0.07       0
  473.36     0.1       0  683.36    0.08       0  793.36    0.06       0
  863.36    0.08       0
#XS Ineff= 2 , 0
                           559.2          2851.7
Permanent Ineff=
       F       F
Bank Sta=281,311.3
XS Rating Curve= 0 ,0
Exp/Cntr(USF)=0,0
Exp/Cntr=0.3,0.1

Type RM Length L Ch R = 1 ,2812    ,210.7,210.7,210.7
XS GIS Cut Line= 3
2333421.72528786656097.0347601782334010.23253103656001.644206301
2334282.46001076656136.265933307
#Sta/Elev= 30
       0 2862.89   124.1 2852.44   156.5 2852.04   197.3 2850.11   229.4 2849.81
     274 2846.28   419.9 2843.01   436.1 2840.93   444.2 2839.22   452.3 2839.02
   456.3 2839.06   462.3 2840.92   468.5 2842.76   500.7 2843.16   569.8 2846.37
   598.4 2845.62   631.2 2845.94     669 2845.05   674.9 2844.24   718.8 2846.19
   739.5 2844.41   749.6 2845.82   799.2 2846.88   808.1 2848.24   821.5 2848.66
   830.4 2849.59   845.1 2853.61     860 2854.06   879.5 2853.22   899.9 2857.12
#Mann= 10, -1 ,  0
       0    0.05       0     100    0.06       0     200    0.05       0
     400    0.08       0   436.1   0.045       0   462.3    0.08       0
     500    0.05       0     510     0.1       0  706.19    0.08       0
  856.19    0.07       0
#XS Ineff= 2 , 0
                          618.43         2849.62
Permanent Ineff=
       F       F
Bank Sta=436.1,462.3
XS Rating Curve= 0 ,0
Exp/Cntr=0.3,0.1

Type RM Length L Ch R = 1 ,2601    ,275.8,275.8,275.8
XS GIS Cut Line= 3
2333500.94099013656176.6430184122334135.80487052656244.801152033
2334360.72784496656241.362719441
#Sta/Elev= 30
       0 2857.71    19.3 2851.25    27.4 2849.91   123.9 2847.53   172.2 2846.91
   208.4 2845.38   241.9 2844.64   389.5 2842.55   405.6 2841.58   417.6 2841.75
  423.78 2840.67   429.7 2839.06   433.7 2838.66   441.8 2839.43   446.6 2840.67
   457.8 2842.78     486 2843.62   518.2 2843.33   538.3 2843.94   622.8 2844.45
   654.9 2845.82     670 2847.26   698.9 2849.07   726.9 2852.58   742.9 2853.45
   754.9 2856.17   774.9 2858.25   806.9 2862.61   846.5 2868.81   863.5 2872.22
#Mann= 7, -1 ,  0
       0    0.07       0      20    0.05       0  423.78   0.045       0
   446.6    0.05       0     610    0.07       0  708.51    0.05       0
  808.51     0.1       0
Bank Sta=423.78,446.6
XS Rating Curve= 0 ,0
Exp/Cntr(USF)=0,0
Exp/Cntr=0.3,0.1

Type RM Length L Ch R = 1 ,2325    ,527.2,527.2,527.2
XS GIS Cut Line= 3
2333419.55355324656455.0374101962334081.07858655 656492.57005486
 2334404.1320802656502.861273017
#Sta/Elev= 30
       0 2860.32    36.7  2853.1   188.4 2846.66   196.9 2846.97   269.1 2844.38
   380.7 2842.59   405.3 2840.37   413.3 2837.74   419.7  2837.7   425.3 2837.83
   432.12840.367   457.4 2841.66   553.5 2842.21   665.2 2844.24   697.7 2843.68
   713.7 2845.27   757.7 2846.48   773.7 2847.93   789.7 2848.52   821.3 2852.14
   837.8 2853.08   865.8 2857.32   889.8 2858.37   905.8 2861.29   933.9 2864.41
   949.8 2867.64   965.8 2868.59   973.8 2872.03   977.8 2873.04   985.8 2873.23
#Mann= 4, -1 ,  0
       0    0.05       0   405.3   0.045       0   432.1    0.05       0
  792.59    0.06       0
Bank Sta=405.3,432.1
XS Rating Curve= 0 ,0
Exp/Cntr(USF)=0,0
Exp/Cntr=0.3,0.1

Type RM Length L Ch R = 1 ,1798    ,305.8,305.8,305.8
XS GIS Cut Line= 2
2333267.57662065656907.5141867812334106.90377111 656731.35910582
#Sta/Elev= 30
       0 2893.65    12.9  2887.3    28.8  2882.2      43    2876    61.9 2868.71
    82.4 2862.92    90.5  2857.6     111 2857.46   115.1 2856.78   123.2 2854.13
     141 2851.82     160 2850.45   200.9 2849.09   222.1  2847.4   233.6 2845.45
   249.9 2845.58   258.1 2847.41   266.3 2847.88   279.5 2844.82   286.7 2842.39
   291.32839.466   294.9    2837     299 2836.81   311.2 2836.91   326.8 2839.79
   352.1 2840.42     442 2840.35   711.8 2842.59   785.3 2844.09   857.6 2844.35
#Mann= 6, -1 ,  0
       0     0.1       0      30    0.06       0     150    0.07       0
   291.3   0.045       0   326.8    0.07       0     460    0.05       0
Bank Sta=291.3,326.8
XS Rating Curve= 0 ,0
Exp/Cntr(USF)=0,0
Exp/Cntr=0.3,0.1

Type RM Length L Ch R = 1 ,1492    ,253.1,253.1,253.1
XS GIS Cut Line= 2
2333276.95156032657259.4862291052334187.77694952656948.624321527
#Sta/Elev= 30
       0 2867.09    33.6 2864.72    49.9 2864.17    66.8 2863.01      80 2860.19
    96.4  2859.1   118.6 2858.53   206.3  2854.4   253.3 2852.82   306.9  2849.8
   328.9 2848.06     388 2842.32   420.3 2839.85   423.5 2839.17   426.1 2838.12
   430.3 2836.47   434.5 2836.34   447.2 2836.41   453.1 2837.99   455.6 2838.45
   476.8 2839.37   539.6 2839.62   650.3 2841.65   700.8 2841.84   763.8  2843.6
   782.7 2843.23   848.7 2843.68   878.3    2845   903.7 2844.77   962.4    2846
#Mann= 10, -1 ,  0
       0     0.1       0      50    0.06       0     150    0.05       0
   426.1   0.045       0   453.1    0.05       0     460    0.07       0
     500    0.05       0     770    0.06       0     810    0.05       0
     880    0.06       0
Bank Sta=426.1,453.1
XS Rating Curve= 0 ,0
Exp/Cntr(USF)=0,0
Exp/Cntr=0.3,0.1

Type RM Length L Ch R = 1 ,1239    ,68.7,68.7,68.7
XS GIS Cut Line= 4
2333348.44979906 657461.546469032333697.30798413657359.004739318
2333747.15038436657324.7762326832334128.91996168657047.877587728
#Sta/Elev= 30
       0  2883.5    15.5 2878.97    19.4 2877.35    33.1 2870.39    49.7 2859.36
    53.9 2858.19    74.8 2858.07   161.2 2850.91   241.5 2851.02   264.3 2850.45
   274.9 2849.62   299.9 2845.84   349.9 2843.23   375.6 2839.62     3872836.965
   391.4 2835.61   401.5 2835.31   410.8 2835.48   415.22837.024   420.5 2839.63
   424.5 2840.59   430.3 2841.55   445.1 2842.46   457.5 2841.83   470.4 2840.44
   484.6 2840.01   539.2 2839.83   613.6 2841.44   682.3 2841.38   895.7 2844.02
#Mann= 11, -1 ,  0
       0     0.1       0      70    0.06       0     180    0.07       0
     240    0.05       0     280    0.08       0     387   0.045       0
   415.2    0.08       0  474.08    0.07       0  504.08    0.06       0
  644.08    0.05       0  744.08    0.06       0
Bank Sta=387,415.2
XS Rating Curve= 0 ,0
Exp/Cntr(USF)=0,0
Exp/Cntr=0.3,0.1

Type RM Length L Ch R = 1 ,1170    ,248.4,248.4,248.4
XS GIS Cut Line= 4
2333398.15294288657503.8922261242333728.85341106657430.728405732
2333805.91930187657355.6135501292334153.20356933657088.321726296
#Sta/Elev= 30
       0 2878.35     6.2 2875.67    18.5 2868.58    30.7 2859.49    34.8 2857.58
    59.4  2857.5    63.5 2855.57    67.7 2851.52    71.7 2850.04    91.2 2851.92
   116.8 2850.39   157.7 2849.65     220 2847.08     269 2845.82   284.7 2844.33
     320 2843.19   370.4 2841.87   376.1 2840.67  383.54 2836.52   387.4 2834.96
   392.5 2834.69   409.7 2836.58   432.7    2838   581.5 2840.58   600.8 2840.17
   661.2 2842.06   726.8 2842.31   740.6  2843.3   786.2 2844.24   884.6  2843.2
#Mann= 11, -1 ,  0
       0     0.1       0      20    0.06       0     120    0.07       0
     220    0.08       0     320    0.06       0  383.54   0.045       0
   409.7    0.08       0  456.31    0.07       0  546.31    0.06       0
  826.31    0.05       0  876.31    0.06       0
Bank Sta=383.54,409.7
XS Rating Curve= 0 ,0
Exp/Cntr(USF)=0,0
Exp/Cntr=0.3,0.1

Type RM Length L Ch R = 1 ,922     ,258.6,258.6,258.6
XS GIS Cut Line= 2
2333410.62218058 657660.49808988 2334228.1889975657489.524040712
#Sta/Elev= 30
       0 2912.34    44.7 2884.73    50.6 2879.75    58.8 2870.15    62.9 2868.81
    79.2 2867.84    87.4 2861.65    91.5 2859.75   103.7 2850.45   111.9 2844.89
     119  2843.3   128.3 2844.87   152.7  2843.5     210 2842.28   234.5 2840.94
   250.9 2841.06   267.2 2840.01   352.2 2838.44   479.7  2837.3   487.9 2836.79
   496.1 2835.28   504.3 2834.43   516.5 2834.25   524.7 2834.25   530.42835.213
   545.4 2837.55   594.1 2838.82     635 2842.03   724.9 2841.42   835.3 2843.31
#Mann= 7, -1 ,  0
       0     0.1       0      10    0.06       0     110    0.05       0
   496.1   0.045       0   530.4    0.05       0     610    0.06       0
     710    0.05       0
Bank Sta=496.1,530.4
XS Rating Curve= 0 ,0
Exp/Cntr(USF)=0,0
Exp/Cntr=0.3,0.1

Type RM Length L Ch R = 1 ,663     ,344.8,344.8,344.8
XS GIS Cut Line= 4
2333386.43624484657835.2942287912333747.37775877657721.483841516
2333889.36976575657757.2528203742334120.24226565657656.449334501
#Sta/Elev= 30
       0 2951.52    22.8 2938.86    39.6 2932.82    60.5  2919.1    76.4 2910.87
    85.7 2903.42    98.7  2889.9   102.5  2886.8   106.7 2885.39   123.5 2884.51
   127.6 2882.98     140 2873.78   165.4 2856.34   190.6 2840.72   203.1 2836.73
   219.9 2838.19   316.4 2836.41   375.1 2836.67   411.8 2835.16   424.7 2833.69
   440.52834.866   474.2 2837.25   490.3 2836.54   548.3 2837.09   565.1 2836.05
   615.2 2837.69   663.3 2837.39   702.5 2838.35   730.6 2841.23   776.8 2841.87
#Mann= 9, -1 ,  0
       0     0.1       0      30    0.06       0     140     0.1       0
     160    0.07       0     240    0.05       0   411.8   0.045       0
   440.5    0.05       0  654.89    0.06       0  764.89    0.05       0
Bank Sta=411.8,440.5
XS Rating Curve= 0 ,0
Exp/Cntr(USF)=0,0
Exp/Cntr=0.3,0.1

Type RM Length L Ch R = 1 ,318     ,211.7,211.7,211.7
XS GIS Cut Line= 3
 2333407.5135615658005.5548072912333861.37194656657930.947949472
2334144.25628246657744.430804926
#Sta/Elev= 30
       0 2952.73    16.9 2943.24    45.3 2929.89    61.5 2919.96    69.6 2913.45
    77.7 2903.49    81.7  2899.9    85.8 2897.99   106.1 2897.03   110.1 2895.04
   138.5 2872.59   154.7 2861.46   162.8 2853.43   166.9 2850.06     179 2842.27
   187.1 2835.93   189.5 2834.78   192.4 2833.82   211.5 2832.48   215.5 2832.99
   220.2 2834.62   300.3 2835.73   349.6 2835.69   397.9 2834.62   458.7 2836.09
   483.5 2835.44   557.6 2837.28     594 2836.96   702.7 2839.78   798.8 2840.08
#Mann= 6, -1 ,  0
       0     0.1       0     110    0.06       0     130     0.1       0
   189.5   0.045       0   220.2    0.05       0  719.95    0.06       0
Bank Sta=189.5,220.2
XS Rating Curve= 0 ,0
Exp/Cntr(USF)=0,0
Exp/Cntr=0.3,0.1

Type RM Length L Ch R = 1 ,107     ,,,
XS GIS Cut Line= 3
2333357.77565629658254.244333353  2333920.435709 658101.92199864
2334265.49242641 657800.38594829
#Sta/Elev= 30
       0  2909.2     2.5 2907.95      36 2904.73    56.4 2895.36    77.8 2888.63
    97.8  2880.6   111.2 2876.61   138.3 2871.43   157.2 2866.87     189 2856.79
   197.3  2852.8   208.3 2850.26   238.7 2836.07   255.3  2833.9   280.3 2834.68
   293.1 2833.27   317.4 2833.76   329.9 2831.49   338.7 2831.41   345.2 2831.98
   350.6 2833.73   374.6 2835.24   408.6 2834.98   437.6 2835.79   549.5 2836.55
   608.4 2834.72   662.6 2836.65   719.3 2836.13   855.4 2838.53  1041.2 2839.74
#Mann= 6, -1 ,  0
       0    0.06       0     170    0.12       0   317.4   0.045       0
   350.6    0.12       0     370    0.05       0  962.91    0.06       0
Bank Sta=317.4,350.6
XS Rating Curve= 0 ,0
Exp/Cntr(USF)=0,0
Exp/Cntr=0.3,0.1
LCMann Table=0

Chan Stop Cuts=-1
Use User Specified Reach Order=0
Composite Channel Slope=5
